HEC-RAS study RICHCK.prj: RICHCK

--- RICHCK.g01 (geometry) --- (continued)

Type RM Length L Ch R = 1 ,44214.3 ,497.6,498.1,496
XS GIS Cut Line= 3
     2054352.798      157106.821     2054415.732      157388.939
     2053992.555      158066.023
#Sta/Elev= 30
       0 1902.19    22.7 1900.59    35.7 1896.34    71.4 1890.36  105.061879.478
   113.7 1875.85   126.7 1867.85   146.2 1867.37   168.9  1858.9  187.941856.864
  285.241854.852   351.2  1854.5  379.481851.857  440.931852.393   514.8 1850.88
   524.7 1848.46   537.1 1850.88  614.381852.482   662.1 1855.84     721 1872.25
   848.6 1891.34   871.5 1891.98   943.5 1889.48   946.8 1888.74  959.121880.974
   966.4 1878.86  998.131879.177 1034.65 1884.57 1063.621885.097  1087.5 1885.18
#Mann= 13 ,-1 , 0
       0     .06       0  105.06     .12       0  187.94     .06       0
  285.24     .12       0  379.48     .06       0  440.93     .12       0
   514.8    .045       0   537.1     .12       0  614.38     .06       0
  959.12    .016       0  998.13     .08       0 1034.65    .016       0
 1063.62     .06       0
#XS Ineff= 2 , 0
                          632.22          1868.5
Permanent Ineff=
       F       F
Bank Sta=514.8,537.1
XS Rating Curve= 0 ,0
Exp/Cntr=0.3,0.1

Type RM Length L Ch R = 1 ,43716.2 ,485.4,487.2,487.4
XS GIS Cut Line= 2
     2054124.933      156980.953     2053658.353      157792.585
#Sta/Elev= 30
       0 1965.59     6.6 1965.98    16.4 1965.47    32.7 1962.65    42.6 1960.18
    68.7 1950.56    94.9 1938.33   117.8 1925.94   147.3 1912.93   166.9 1902.58
   186.6 1889.58   209.5 1871.94   232.4 1856.81   248.8 1849.77   258.6 1849.03
   266.8 1847.51   278.2 1846.56   284.8 1847.73   291.3 1849.03   304.4 1849.25
   330.6 1848.77   340.4 1849.64   353.5 1848.85  377.951848.943   513.9 1850.13
   536.8 1851.08   576.1 1854.07   618.7 1855.02   821.6 1863.83   936.2 1867.93
#Mann= 4 ,-1 , 0
       0     .12       0   266.8    .045       0   284.8     .12       0
  377.95     .06       0
Bank Sta=266.8,284.8
XS Rating Curve= 0 ,0
Exp/Cntr=0.3,0.1

Type RM Length L Ch R = 1 ,43229   ,452.2,456.1,455.3
XS GIS Cut Line= 2
     2053701.756       156776.96     2053194.371      157577.343
#Sta/Elev= 30
       0 1934.52    13.1 1928.54    42.6 1916.67    55.7 1910.44    62.3 1909.53
    78.7 1909.28   114.8 1902.84   121.3 1901.03   131.2 1899.51   134.4 1898.53
   144.3 1893.35   157.4 1888.03   180.4 1876.58   229.5  1848.6   232.8 1847.31
   245.9  1845.5     254 1845.55   262.3 1844.38   272.2 1844.86   275.4 1845.55
   278.7 1846.29   288.6 1846.82   301.7 1845.82  327.111846.664     423 1847.92
   580.4 1851.93   649.3 1855.37   744.4 1858.76   836.2 1863.71   947.7 1867.52
#Mann= 4 ,-1 , 0
       0     .12       0     254    .045       0   275.4     .12       0
  327.11     .06       0
Bank Sta=254,275.4
XS Rating Curve= 0 ,0
Exp/Cntr=0.3,0.1

Type RM Length L Ch R = 1 ,42772.9 ,132.8,133.8,134.1
XS GIS Cut Line= 3
     2053847.155      156002.221      2053298.11      156644.582
     2052848.892      157204.478
#Sta/Elev= 30
       0 1869.19    98.3 1879.58   117.9  1880.5   209.6  1877.2   268.6 1883.57
   301.3 1889.52   379.9 1896.72   425.8 1896.49   458.5 1894.41   501.1 1899.72
   533.9 1899.74   681.3 1888.35     750 1888.57     773 1886.52   795.9  1881.2
   835.2 1868.34   877.8 1856.75   887.6 1852.41   897.5 1843.72   907.3 1842.04
     914 1843.47   933.5 1844.89 1014.941845.479  1143.3 1844.99  1310.5 1846.83
  1346.5 1850.57  1412.1 1864.24  1444.9 1868.72  1510.4 1873.93  1562.9 1874.16
#Mann= 4 ,-1 , 0
       0     .12       0   897.5    .045       0     914     .12       0
 1014.94     .06       0
Bank Sta=897.5,914
XS Rating Curve= 0 ,0
Exp/Cntr=0.3,0.1

Type RM Length L Ch R = 1 ,42639.1 ,760,741.8,711.4
XS GIS Cut Line= 4
     2053745.159      155969.669      2053289.43       156455.78
      2052831.53      156991.804     2052838.041      157184.946
#Sta/Elev= 30
       0 1848.18    88.2 1846.69  213.391846.576     294 1849.59   431.2 1847.27
  536.311848.198   646.7 1848.02  737.221844.833     774 1844.54     850    1844
   858.8 1843.04   866.4  1842.2   873.8 1842.97   879.5 1844.34  887.261843.974
     968 1844.37  1053.2 1842.93  1135.2 1844.08  1292.6 1843.88  1371.3 1845.92
 1391.791847.575  1400.8 1848.45  1413.9 1851.95  1433.5 1852.88 1447.541856.867
  1456.5 1858.48  1472.8 1864.08  1495.8 1868.36  1525.2 1871.54  1564.6 1873.67
#Mann= 10 ,-1 , 0
       0     .06       0  213.39    .016       0  536.31     .06       0
  737.22     .12       0     774     .06       0   858.8    .045       0
   873.8     .08       0  887.26     .06       0 1391.79    .016       0
 1447.54     .06       0
#XS Ineff= 2 , 0
          726.29 1851.62 1247.26          1855.5
Permanent Ineff=
       F       F
Bank Sta=858.8,873.8
XS Rating Curve= 0 ,0
Exp/Cntr=0.3,0.1

Type RM Length L Ch R = 1 ,41897.3 ,175.7,174.2,173.3
XS GIS Cut Line= 4
     2053158.787      155800.398     2052686.131      156258.297
     2052805.489      156996.144     2052811.999      157178.436
#Sta/Elev= 30
       0  1885.8   101.5 1895.97   173.5 1897.05   271.8 1885.63   363.4 1867.93
   389.6 1868.46   445.3 1874.67   497.7  1884.5   658.1 1928.26   720.4 1932.46
   772.8  1927.2   844.9 1909.22   867.9 1900.44   890.8 1886.21   910.5 1878.21
  939.08 1861.83   966.2 1847.16   982.6 1840.99  1011.3 1838.86  1015.4 1838.16
  1031.8 1839.39 1032.851839.839  1041.6 1842.05  1343.2  1842.7 1442.391848.388
  1460.9 1853.04  1483.7 1854.24 1499.571860.875    1526 1866.51  1587.9  1872.2
#Mann= 7 ,-1 , 0
       0     .06       0  939.08     .12       0  1011.3    .045       0
  1031.8     .12       0 1032.85     .06       0 1442.39    .016       0
 1499.57     .06       0
Bank Sta=1011.3,1031.8
XS Rating Curve= 0 ,0
Exp/Cntr=0.3,0.1

Type RM Length L Ch R = 1 ,41723.1 ,493.1,493.3,490.1
XS GIS Cut Line= 3
     2052407.044      155950.342     2052574.221      156618.025
      2052702.58      157317.931
#Sta/Elev= 30
       0 1994.61    81.9 1995.81   245.8 1982.29   317.9 1984.31   370.4 1980.63
   416.2 1971.55   442.5  1963.8   462.1 1956.77   481.8 1946.52   511.3  1934.8
  531.611923.725  589.451888.103   655.5  1845.3   665.4 1840.48   680.8 1838.34
   694.8 1837.77   701.4 1838.68   717.8 1841.07  908.781840.073   924.4 1841.77
   956.1 1841.67  1144.1 1843.34  1183.4 1847.48 1222.951857.123  1252.3  1857.9
  1265.4 1863.54 1269.861863.606    1314 1861.78 1398.561862.542  1399.9 1862.55
#Mann= 11 ,-1 , 0
       0     .06       0  531.61     .12       0  589.45     .06       0
   680.8    .045       0   701.4     .06       0  908.78     .12       0
   956.1     .06       0 1222.95    .016       0 1269.86     .06       0
    1314     .12       0 1398.56     .06       0
Bank Sta=680.8,701.4
XS Rating Curve= 0 ,0
Exp/Cntr=0.3,0.1

Type RM Length L Ch R = 1 ,41229.8 ,302.2,305.2,305.5
XS GIS Cut Line= 2
     2052134.916      156117.238     2052213.041      157373.748
#Sta/Elev= 30
       0 2020.48      23  2013.4    42.6 2005.42    75.4 1993.82   111.5 1982.75
   163.9 1957.02     236 1929.64   255.7 1920.13   268.8 1915.02     318 1898.08
   383.6  1873.7   419.6 1859.46   455.7 1841.78   465.5 1839.84   504.9  1839.2
   511.4 1837.61   514.7 1836.45   527.8 1836.22   537.7 1837.48     541 1838.42
  549.531838.573   583.6 1838.04   613.1 1839.57  1009.8 1841.91  1104.8 1843.43
 1155.411845.392  1173.7 1846.62 1196.481846.511  1222.9 1846.75  1258.9 1849.39
#Mann= 6 ,-1 , 0
       0     .06       0   511.4    .045       0   537.7     .12       0
  549.53     .06       0 1155.41    .016       0 1196.48     .08       0
Bank Sta=511.4,537.7
XS Rating Curve= 0 ,0
Exp/Cntr=0.3,0.1

Type RM Length L Ch R = 1 ,40924.6 ,492.2,540.7,533
XS GIS Cut Line= 3
     2051946.114      156112.898     2051900.541      156271.318
      2051894.03      157312.985
#Sta/Elev= 30
       0 1992.12    64.6 1970.48   135.8 1951.47   145.4 1950.27   164.8 1944.41
   194.3 1938.98   266.4 1930.86   289.3 1926.62   305.7 1921.38   315.5 1920.19
   351.6 1907.79   367.9 1899.96  387.05 1887.96   413.8 1865.91   436.7 1848.87
   456.4 1837.44   500.41837.169   534.4 1836.14   544.8 1834.98   557.9 1836.86
   567.8  1838.8   803.6 1839.41 1021.561842.078  1049.3 1842.22  1062.4 1841.05
 1070.171843.036  1078.8 1845.53 1141.641847.599 1200.721850.349  1206.5 1850.51
#Mann= 9 ,-1 , 0
       0     .06       0  387.05     .12       0   500.4     .06       0
   534.4    .045       0   557.9     .06       0 1021.56    .016       0
 1070.17     .06       0 1141.64     .08       0 1200.72     .12       0
#XS Ineff= 2 , 0
                          840.47            1862
Permanent Ineff=
       F       F
Bank Sta=534.4,557.9
XS Rating Curve= 0 ,0
Exp/Cntr=0.3,0.1

Type RM Length L Ch R = 1 ,40383.9 ,790.9,744.3,714.6
XS GIS Cut Line= 5
       2051301.8      156212.507     2051488.003       156459.83
     2051513.605      156917.368     2051838.258       157064.07
     2051848.675      157306.257
#Sta/Elev= 30
       0 1950.79    39.1 1944.17    68.4 1938.02    94.5 1930.69   153.2 1911.48
   224.8 1883.63   237.9 1880.04     277 1865.63   306.3 1857.68   355.4 1850.15
   404.5  1839.5   440.5 1836.75   450.3  1833.9  489.71 1835.03   499.4 1834.41
   509.2 1833.86   519.1  1834.5  534.751836.483   633.6 1838.58   761.3 1837.81
   888.8 1838.37  1156.8 1842.08 1162.811841.419  1186.3 1841.75    1206  1840.5
 1210.321841.323  1228.9 1844.11 1255.011845.147 1298.721846.144  1366.5 1849.11
#Mann= 9 ,-1 , 0
       0     .06       0  489.71     .07       0   499.4    .045       0
   519.1     .07       0  534.75     .06       0 1162.81    .016       0
 1210.32     .06       0 1255.01     .08       0 1298.72     .06       0
#XS Ineff= 2 , 0
                          658.24         1862.98
Permanent Ineff=
       F       F
Bank Sta=499.4,519.1
XS Rating Curve= 0 ,0
Exp/Cntr=0.3,0.1

Type RM Length L Ch R = 1 ,39639.6 ,112.2,101.4,93.3
XS GIS Cut Line= 4
     2050632.746      156282.603     2050654.447      156545.189
     2051811.565      157074.269     2051818.076      157321.665
#Sta/Elev= 30
       0 1862.17   20.611861.649    65.1 1859.36   84.521857.336   221.2 1846.96
   263.5 1844.75  317.291844.964  323.071844.914   338.9 1844.29   355.3 1840.99
   381.5 1840.37  390.891838.648   397.9 1837.44  420.511836.948  457.421835.105
   479.9 1834.43   496.3 1831.04   502.9 1830.62   525.8 1831.35   571.7 1835.02
   594.7 1834.61    1385 1838.93 1551.521841.329  1578.2 1841.64  1594.4 1840.52
 1599.821841.272  1607.5 1842.63  1623.7 1843.82  1679.1 1845.19  1783.3 1849.31
#Mann= 12 ,-1 , 0
       0     .06       0   20.61    .016       0   84.52     .06       0
  317.29    .016       0  323.07     .08       0  390.89     .06       0
  420.51     .08       0  457.42     .06       0   496.3    .045       0
   525.8     .06       0 1551.52    .016       0 1599.82     .06       0
Bank Sta=496.3,525.8
XS Rating Curve= 0 ,0
Exp/Cntr=0.3,0.1

Type RM Length L Ch R = 1 ,39538.2 ,300.6,302,303.6
XS GIS Cut Line= 4
     2050576.322      156286.943     2050621.895      156629.825
     2051750.801      157139.373     2051757.312      157386.769
#Sta/Elev= 30
       0 1862.16   45.761859.994   75.561857.987  129.421853.565  138.731853.275
  182.771849.825   241.5 1846.71  248.791845.002   254.5 1843.11  307.631842.413
   331.71841.667  343.761841.721  408.661840.224  441.071838.143   463.9 1835.36
  533.791834.692   558.9  1835.8  574.171831.707   581.8 1830.56   588.4 1830.39
   611.3 1830.86   651.81834.508   804.6 1836.18  1260.1 1837.25  1482.9 1839.84
 1542.961841.738 1575.361842.431 1604.581842.694  1753.8 1846.96    1832 1853.68
#Mann= 20 ,-1 , 0
       0     .06       0   45.76     .12       0   75.56    .016       0
  129.42     .06       0  138.73     .08       0  182.77     .06       0
  248.79    .016       0  307.63     .12       0   331.7     .08       0
  343.76     .12       0  408.66    .016       0  441.07     .06       0
  533.79     .12       0  574.17     .06       0   581.8    .045       0
   611.3     .12       0   651.8     .06       0 1542.96     .08       0
 1575.36     .12       0 1604.58     .06       0
Bank Sta=581.8,611.3
XS Rating Curve= 0 ,0
Exp/Cntr=0.3,0.1

Type RM Length L Ch R = 1 ,39236.2 ,504.5,513.2,518.7
XS GIS Cut Line= 3
     2050127.755      156689.597     2051451.322      157386.769
     2051438.301       157547.36
#Sta/Elev= 30
       0 1931.84    62.3 1930.46   177.2 1922.72   337.9 1908.93   416.6 1898.64
   446.2 1893.02   475.7 1882.96   534.7 1856.66  564.091837.491  597.691834.924
  656.531831.976   660.9 1830.92   679.1 1830.02   685.6 1830.88  689.911831.785
   711.9 1831.76   731.6 1834.55   859.5  1833.7  1151.5 1835.34 1418.88 1841.69
  1499.2 1846.92    1525 1846.13  1534.6 1851.24  1557.2 1870.62 1564.26 1871.94
  1573.3 1870.36  1593.9 1870.74 1623.54 1872.32  1634.5 1877.96  1657.1 1881.17
#Mann= 11 ,-1 , 0
       0     .06       0  564.09    .016       0  597.69     .06       0
  656.53     .08       0   660.9    .045       0   685.6     .08       0
  689.91     .06       0 1418.88     .12       0 1564.26     .08       0
  1593.9    .016       0 1623.54     .06       0
Bank Sta=660.9,685.6
XS Rating Curve= 0 ,0
Exp/Cntr=0.3,0.1

Type RM Length L Ch R = 1 ,38722.9 ,368.1,374.1,376.3
XS GIS Cut Line= 2
     2050040.388      156850.084     2051043.336      157888.071
#Sta/Elev= 30
       0    1911    16.4 1905.91    45.9 1900.98    68.9 1898.77   124.6 1898.72
   154.2 1897.28   177.1 1894.78  214.931886.858   229.6 1882.57   255.9 1872.18
   295.2 1848.91   311.6 1841.84   341.2  1834.9  387.571833.687  834.111830.757
   849.6 1829.37   862.7 1828.98   868.7 1830.05  876.621831.632   980.8  1832.5
  1020.2 1835.56  1180.9 1856.12  1226.9  1864.7  1244.41869.583  1253.1 1873.26
  1276.1 1873.92 1283.541878.009  1292.5 1882.69  1394.2 1911.01  1443.4 1925.88
#Mann= 9 ,-1 , 0
       0     .06       0  214.93     .12       0  387.57     .06       0
  834.11     .08       0   849.6    .045       0   868.7     .08       0
  876.62     .06       0  1244.4    .016       0 1283.54     .06       0
Bank Sta=849.6,868.7
XS Rating Curve= 0 ,0
Exp/Cntr=0.3,0.1

Type RM Length L Ch R = 1 ,38348.9 ,630.9,631.2,625.3
XS GIS Cut Line= 3
     2049884.048      156998.748     2050622.329       158024.79
     2050814.603      158182.776
#Sta/Elev= 30
       0 1894.61      36 1880.73    91.7 1870.25   160.5 1862.74   242.3  1864.2
     262 1861.32   275.1 1857.34  287.861851.537   314.4 1837.96   327.5  1832.7
   348.91831.743   481.4 1831.62   566.5 1829.82  813.43 1831.08     822 1831.21
   831.8 1828.42   844.9 1827.72   853.8 1828.47   871.1 1830.47   910.4 1830.36
  933.091835.687   985.7  1840.1  1129.8 1856.65 1161.341861.776  1169.1 1864.12
  1195.3 1865.07 1200.991867.017    1251 1874.48  1332.8 1893.83  1512.9 1930.08
#Mann= 9 ,-1 , 0
       0     .06       0  287.86     .12       0   348.9     .06       0
  813.43     .12       0   831.8    .045       0   853.8     .12       0
  933.09     .06       0 1161.34    .016       0 1200.99     .12       0
Bank Sta=831.8,853.8
XS Rating Curve= 0 ,0
Exp/Cntr=0.3,0.1

Type RM Length L Ch R = 1 ,37717.6 ,793,792,781.8
XS GIS Cut Line= 3
     2049432.659      157159.339     2050279.881       158020.45
     2050693.076      158148.922
#Sta/Elev= 30
       0 1940.67   14.741934.269    58.9 1916.54    85.1 1908.73   173.5 1888.13
   297.9  1864.1   343.7 1850.73   389.6 1843.27   422.3 1829.22   569.6 1828.25
   717.91829.568   743.1 1827.51   762.8 1826.46   772.6  1827.7   785.7  1829.7
  1057.4 1831.35  1149.1 1838.97 1198.09 1847.24 1219.69 1852.39  1244.1 1862.05
  1283.4 1864.31 1296.811870.271  1306.4 1874.56  1368.6 1886.65  1401.4 1895.37
    1444 1902.59  1486.6 1904.27  1601.4 1903.32    1621 1901.55  1640.7 1905.68
#Mann= 8 ,-1 , 0
       0     .12       0   14.74     .06       0   717.9     .12       0
   743.1    .045       0   772.6     .06       0 1198.09     .12       0
 1219.69    .016       0 1296.81     .12       0
Bank Sta=743.1,772.6
XS Rating Curve= 0 ,0
Exp/Cntr=0.3,0.1

Type RM Length L Ch R = 1 ,36925.7 ,1604.9,1629.7,1550
XS GIS Cut Line= 3
     2049148.805      157420.623      2050016.86      158288.679
     2050424.846      158319.061
#Sta/Elev= 30
       0 1951.01  124.051891.985     180 1868.39   222.6 1851.83   242.2 1846.04
     275 1841.29   353.6 1835.23   405.9 1829.06  478.531828.363   487.8 1825.69
   500.9 1824.16   517.2 1825.23  524.361826.401  527.031826.546  601.961827.509
  1045.1 1829.13  1093.4 1829.77 1188.541834.568  1227.6 1834.26 1239.941835.814
    1280 1842.63 1289.421846.089  1299.6  1848.1  1328.51847.785  1338.9 1852.27
  1355.3 1854.91  1404.4  1869.5  1456.7 1887.02  1515.6 1903.45  1636.7 1932.38
#Mann= 13 ,-1 , 0
       0     .12       0  124.05     .06       0  478.53     .12       0
   487.8    .045       0   517.2     .12       0  524.36     .06       0
  527.03     .12       0  601.96     .06       0  1045.1     .12       0
 1188.54     .06       0 1239.94     .12       0 1289.42    .016       0
  1328.5     .12       0
#XS Ineff= 2 , 0
                         1005.31         1847.33
Permanent Ineff=
       F       F
Bank Sta=487.8,517.2
XS Rating Curve= 0 ,0
Exp/Cntr=0.3,0.1

Type RM Length L Ch R = 1 ,35296   ,1110.4,1117.4,1114.6
XS GIS Cut Line= 2
     2048967.291      157593.942     2048905.749      159169.755
#Sta/Elev= 30
       0 1858.67    26.2  1850.7    62.3 1843.56   131.1 1833.86   268.8 1827.77
   472.1  1824.4   744.2 1825.31   763.9    1824     918 1824.86   934.4 1823.91
   947.5 1821.89   956.7 1823.92   967.2 1825.09  1029.5 1824.75  1039.3 1826.56
  1052.4 1831.88  1065.6 1832.86 1071.541834.701  1098.3 1835.17 1102.27 1837.62
  1108.2 1841.75  1131.1 1846.16    1200 1852.56 1230.881854.421 1315.181859.081
 1382.491865.085 1383.741865.237  1416.4 1868.01  1462.3 1869.16    1577 1868.64
#Mann= 9 ,-1 , 0
       0     .06       0   934.4    .045       0   956.7     .06       0
 1071.54    .016       0 1102.27     .06       0 1230.88     .08       0
 1315.18     .06       0 1382.49     .08       0 1383.74     .06       0
Bank Sta=934.4,956.7
XS Rating Curve= 0 ,0
Exp/Cntr=0.3,0.1

Type RM Length L Ch R = 1 ,34178.6 ,462.4,466.9,452.7
XS GIS Cut Line= 3
     2048588.909      157468.366     2048454.331      157660.069
     2048224.326      159017.846
#Sta/Elev= 30
       0 1899.42   169.2 1865.56   191.9 1858.97   250.6 1836.97   260.5  1835.4
   276.8 1829.56   286.7 1827.42   309.6 1824.92   493.2  1824.3     572 1825.35
   712.9 1823.24   844.1 1824.64     890 1824.17   916.2 1821.77  1024.4 1822.67
  1033.2  1820.9  1040.8 1819.11  1060.5 1821.59  1076.9 1823.08 1083.43 1825.07
    1090 1829.12 1104.491830.296    1113 1830.44  1129.4  1845.1 1135.981847.473
  1162.1 1854.02  1204.8 1856.54  1434.3 1878.75    1572 1897.96  1611.3 1905.06
#Mann= 6 ,-1 , 0
       0     .06       0  1033.2    .045       0  1060.5     .12       0
 1083.43    .016       0 1104.49     .08       0 1135.98     .06       0
Bank Sta=1033.2,1060.5
XS Rating Curve= 0 ,0
Exp/Cntr=0.3,0.1

Type RM Length L Ch R = 1 ,33711.7 ,550.4,558,562.6
XS GIS Cut Line= 2
     2048371.895       157372.88     2047783.333      159030.324
#Sta/Elev= 30
       0 1884.35    26.2 1880.64    98.3 1865.86   170.3 1846.85  217.171837.334
  236.561834.945   268.6 1830.49   294.8 1824.64   311.2 1823.79   550.2 1824.75
   989.1 1823.56    1071 1821.73  1080.8 1820.29  1090.7  1818.8  1100.5 1820.34
  1110.3 1821.69 1123.841829.449  1133.3 1835.36 1152.58 1835.76    1166 1843.54
 1183.931847.543 1287.491871.736 1298.621874.378  1480.4 1908.26  1595.1 1936.22
  1644.2 1949.74 1674.891956.058 1703.271966.781 1735.411980.046  1758.8 1988.37
#Mann= 13 ,-1 , 0
       0     .06       0  217.17     .08       0  236.56     .06       0
  1080.8    .045       0  1100.5     .08       0 1123.84    .016       0
 1152.58     .08       0 1183.93     .06       0 1287.49     .08       0
 1298.62     .06       0 1674.89     .08       0 1703.27     .06       0
 1735.41     .08       0
#XS Ineff= 2 , 0
          366.31 1849.76
Permanent Ineff=
       F       F
Bank Sta=1080.8,1100.5
XS Rating Curve= 0 ,0
Exp/Cntr=0.3,0.1

Type RM Length L Ch R = 1 ,33153.7 ,491,489,481.2
XS GIS Cut Line= 3
     2048211.305       157203.61     2047464.777      158293.019
     2047451.756      158870.276
#Sta/Elev= 30
       0 1880.09    91.8 1865.01   180.2  1846.4     272 1834.47   350.6 1827.93
   445.7  1824.7   760.3 1820.32  1045.4 1821.86  1071.6 1820.05  1173.2 1820.75
  1186.3 1818.55  1199.4 1817.39    1206 1818.92 1233.091824.703  1238.7 1826.66
  1258.4 1826.73  1261.7 1827.82 1271.181836.004  1284.6 1844.66  1307.5 1854.34
 1368.221872.717    1442 1890.56 1521.22 1912.64  1547.31919.485  1619.2 1940.71
  1648.7 1953.45 1686.911965.792  1733.41982.598  1770.1    1991    1898 2007.31
#Mann= 10 ,-1 , 0
       0     .06       0  1186.3    .045       0    1206     .06       0
 1233.09    .016       0 1271.18     .08       0 1368.22     .06       0
 1521.22     .08       0  1547.3     .06       0 1686.91     .08       0
  1733.4     .06       0
Bank Sta=1186.3,1206
XS Rating Curve= 0 ,0
Exp/Cntr=0.3,0.1

Type RM Length L Ch R = 1 ,32664.6 ,842.5,844.4,839.6
XS GIS Cut Line= 2
     2047625.367      157003.957     2046980.187      158709.979
#Sta/Elev= 30
       0  1862.2      59 1848.88   118.1 1838.65   147.6 1834.71   183.7 1832.66
   564.2 1821.29   734.8 1821.57   836.5  1820.2   879.2 1821.12   905.4 1818.74
  1046.5 1820.48  1121.9 1819.94  1133.8 1817.89  1141.6 1816.51  1154.7 1817.96
 1155.991818.558  1167.8 1825.25  1190.8 1827.42  1197.4 1832.62  1203.9 1839.91
  1208.21842.489  1226.9  1851.5  1246.6 1858.69  1325.3 1882.77  1463.1 1926.97
 1531.081945.981 1570.531956.254 1638.861973.492 1678.851982.419  1823.9 2006.83
#Mann= 9 ,-1 , 0
       0     .06       0  1133.8    .045       0  1154.7     .06       0
 1155.99    .016       0  1208.2     .12       0 1531.08     .06       0
 1570.53     .12       0 1638.86     .08       0 1678.85     .06       0
Bank Sta=1133.8,1154.7
XS Rating Curve= 0 ,0
Exp/Cntr=0.3,0.1

Type RM Length L Ch R = 1 ,31820.3 ,772.2,772.4,770
XS GIS Cut Line= 2
     2047213.041      156826.005     2046705.228      158423.228
#Sta/Elev= 30
       0 1880.73   137.8 1854.23   226.3 1835.19   285.4  1828.6   419.8 1821.38
     492 1819.77   836.4 1818.17   905.2 1818.82   931.5 1816.91   967.6 1817.83
  1003.6 1816.95  1010.2 1815.02  1023.3 1815.69  1026.6 1816.92  1056.1 1818.82
  1164.4 1818.96 1181.44 1820.73  1193.9  1826.2  1210.3 1826.61  1213.6 1827.14
 1217.551829.585  1234.81838.652 1248.551844.009  1295.5 1862.31 1344.121877.174
  1459.5 1913.38    1512  1927.9    1594 1954.83  1649.8 1974.51    1676 1981.36
#Mann= 8 ,-1 , 0
       0     .06       0  1003.6    .045       0  1026.6     .06       0
 1181.44    .016       0 1217.55     .08       0  1234.8     .12       0
 1248.55     .06       0 1344.12     .12       0
Bank Sta=1003.6,1026.6
XS Rating Curve= 0 ,0
Exp/Cntr=0.3,0.1

Type RM Length L Ch R = 1 ,31047.9 ,578.8,577.8,574.6
XS GIS Cut Line= 3
     2046614.082      156548.228     2046162.694      158045.623
     2046227.798      158293.019
#Sta/Elev= 30
       0 1937.74      59 1910.77   160.7 1855.67   252.5 1833.56  325.931828.759
   613.1 1817.64  1055.8  1818.3  1180.3 1814.55  1190.2 1813.26    1200 1814.39
  1262.3 1816.38 1300.411842.486 1333.741841.684  1373.8 1843.17  1390.2 1851.52
  1406.6 1854.51    1423 1862.57  1478.7 1875.12  1498.4 1874.84 1517.751870.529
 1541.781867.619    1564 1862.26  1586.9 1861.25  1629.6 1864.74  1659.1 1872.66
 1729.451873.119  1754.2 1874.31  1773.8 1878.04  1793.5 1886.38  1819.8  1887.9
#Mann= 9 ,-1 , 0
       0     .12       0  325.93     .06       0  1180.3    .045       0
    1200     .12       0 1300.41    .016       0 1333.74     .08       0
 1517.75     .06       0 1541.78     .08       0 1729.45     .06       0
Bank Sta=1180.3,1200
XS Rating Curve= 0 ,0
Exp/Cntr=0.3,0.1

Type RM Length L Ch R = 1 ,30470.1 ,988,988.8,982.5
XS GIS Cut Line= 3
     2045958.701      156457.082     2045680.923      157880.693
     2045772.069       158310.38
#Sta/Elev= 30
       0 1931.99    52.4 1890.87    81.8 1869.71    98.2 1859.05   124.4 1845.31
   144.1 1839.15  209.82 1833.46   288.1 1822.18   363.4 1817.12     645 1816.58
   792.4 1814.64 1068.591816.295  1083.8 1814.74 1102.691815.477  1204.9 1815.99
  1224.5 1813.56  1244.2 1814.17    1254 1812.88  1270.4  1814.8 1277.161817.739
    12861823.056  1303.1 1834.05    1326 1835.01  1335.9 1839.15 1354.141843.067
  1369.51844.801    1457 1853.13  1499.6 1854.22 1676.771865.501  1889.7 1871.29
#Mann= 11 ,-1 , 0
       0     .12       0  209.82     .06       0 1068.59     .12       0
 1102.69     .06       0  1244.2    .045       0  1270.4     .06       0
 1277.16     .12       0    1286    .016       0 1354.14     .06       0
  1369.5    .016       0 1676.77     .06       0
Bank Sta=1244.2,1270.4
XS Rating Curve= 0 ,0
Exp/Cntr=0.3,0.1

Type RM Length L Ch R = 1 ,29481.3 ,1082.7,1452.1,1451.3
XS GIS Cut Line= 2
     2045333.701      156365.936     2045138.388      157967.498
#Sta/Elev= 30
       0 1950.52    19.7 1943.86    55.8 1925.67    75.4 1911.04   118.1 1884.64
   180.4  1837.1   203.3  1824.7   226.3 1816.24   293.21815.154  322.961814.865
  442.951814.242  464.551813.937  577.981814.253   613.2 1815.03   623.1 1811.66
   629.5 1810.49   649.3 1811.56   662.4 1814.27   908.4 1813.56     9811816.191
   990.4 1818.24  1029.7  1835.9 1059.051839.724  1262.5 1856.45 1453.771863.089
    15061863.954 1525.32 1864.46 1569.121865.438 1602.56 1864.83  1613.4 1865.97
#Mann= 15 ,-1 , 0
       0     .12       0   293.2     .06       0  322.96     .08       0
  442.95     .06       0  464.55     .08       0  577.98     .06       0
   623.1    .045       0   649.3     .06       0     981     .12       0
 1059.05     .06       0 1453.77     .12       0    1506     .08       0
 1525.32     .12       0 1569.12    .016       0 1602.56     .08       0
Bank Sta=623.1,649.3
XS Rating Curve= 0 ,0
Exp/Cntr=0.3,0.1

Type RM Length L Ch R = 1 ,28029.2 ,326.5,325.4,324.2
XS GIS Cut Line= 3
     2044808.527      156313.853     2044673.978      156500.485
     2044574.152      157780.866
#Sta/Elev= 30
       0 1972.39    90.7 1997.73   142.6 2008.76   158.8 2010.81     175 2010.75
     188 2008.98   200.9  2005.5   220.4 1997.48   256.3 1977.59     289 1957.24
   357.8 1909.97   367.7 1897.76   380.8 1889.89   397.2 1875.29   439.8 1845.52
   456.1 1832.57     466 1822.86   475.8 1809.57   488.9 1808.52   505.3 1809.43
  555.931812.859   934.5 1814.51    1226 1818.34  1271.9 1821.24  1307.9 1826.39
  1337.4 1832.54  1373.5 1834.39 1402.691837.663 1446.431839.356  1514.3 1844.07
#Mann= 6 ,-1 , 0
       0     .12       0   475.8    .045       0   505.3     .12       0
  555.93     .06       0 1402.69    .016       0 1446.43     .06       0
Bank Sta=475.8,505.3
XS Rating Curve= 0 ,0
Exp/Cntr=0.3,0.1

Type RM Length L Ch R = 1 ,27703.8 ,524.8,528.1,529.4
XS GIS Cut Line= 3
     2044496.027      156253.089     2044345.802      156565.859
     2044274.673      157811.248
#Sta/Elev= 30
       0 2040.42    19.6  2043.2    42.6 2038.65    65.5 2028.31   104.8 2004.33
   160.4 1962.41   193.1 1935.43     216 1919.16   248.8 1891.99   281.5 1862.86
     347 1821.14   363.4 1814.94   379.7 1810.85   451.8 1811.75   474.7 1807.99
   494.3 1807.43   504.1 1807.99     514 1811.36     550 1810.23  577.27 1812.03
   605.6 1813.13   635.1 1812.17   844.6 1812.84  1178.6 1819.16 1318.021823.231
  1348.8 1823.98  1388.1 1827.23 1426.571827.722  1492.9 1827.21  1594.4  1828.7
#Mann= 6 ,-1 , 0
       0     .12       0   474.7    .045       0   504.1     .12       0
  577.27     .06       0 1318.02    .016       0 1426.57     .06       0
Bank Sta=474.7,504.1
XS Rating Curve= 0 ,0
Exp/Cntr=0.3,0.1

Type RM Length L Ch R = 1 ,27175.6 ,1359.5,1363.6,1355.8
XS GIS Cut Line= 3
     2044161.826      156040.415     2043983.874      156201.005
     2043775.541      157628.957
#Sta/Elev= 30
       0  1970.6    48.6 1956.82    97.2 1937.62   171.7 1896.76   239.7 1853.75
   328.2  1817.7   357.8 1811.65     466 1811.31   475.8 1810.11   483.1 1806.85
   492.2 1806.23   505.4 1806.81   511.9 1809.81   521.8 1811.37  567.741810.518
  1338.4 1813.86  1374.5  1818.2 1392.241825.363  1400.7 1827.72 1416.881828.113
    1427 1828.18 1446.731839.694  1453.2 1844.51  1476.2 1851.62  1495.8 1853.64
  1535.2 1853.22 1553.471855.538 1595.991860.003 1630.281867.995  1682.8 1881.59
#Mann= 10 ,-1 , 0
       0     .12       0   483.1    .045       0   505.4     .12       0
  567.74     .06       0 1392.24    .016       0 1416.88     .08       0
 1446.73     .12       0 1553.47    .016       0 1595.99     .06       0
 1630.28     .12       0
Bank Sta=483.1,505.4
XS Rating Curve= 0 ,0
Exp/Cntr=0.3,0.1

Type RM Length L Ch R = 1 ,25812   ,834.4,850.1,862.2
XS GIS Cut Line= 4
     2043849.326      155406.735     2043393.596      155541.283
     2043202.624      157181.908     2043094.117      157329.478
#Sta/Elev= 30
       0 1889.44   114.7  1867.2   147.5 1858.56  186.651842.458     2371823.301
   268.7 1817.76   406.4 1809.95  1055.2 1810.03  1150.3 1807.24  1333.8 1808.96
  1392.8  1805.6 1481.511809.149 1551.621808.587  1609.1 1807.96    1632 1804.88
  1638.6 1804.45  1658.2 1804.87  1677.9 1809.06  1907.3 1812.03  1930.2 1813.15
 1941.331816.742  1949.9 1819.36  1972.8 1819.49 1986.121828.365  2094.1 1879.98
  2133.4 1891.02 2184.051897.777 2251.341910.068 2281.831913.503    2310 1914.04
#Mann= 12 ,-1 , 0
       0     .06       0  186.65     .12       0     237     .06       0
 1481.51     .12       0 1551.62     .06       0    1632    .045       0
  1658.2     .06       0 1941.33    .016       0 1986.12     .12       0
 2184.05     .06       0 2251.34     .08       0 2281.83    .016       0
#XS Ineff= 2 , 0
          969.47 1830.71
Permanent Ineff=
       F       F
Bank Sta=1632,1658.2
XS Rating Curve= 0 ,0
Exp/Cntr=0.3,0.1

Type RM Length L Ch R = 1 ,24961.9 ,651.1,656.6,647.4
XS GIS Cut Line= 3
     2043831.964      155311.248     2043493.423       155332.95
     2042234.742      156713.158
#Sta/Elev= 30
       0 1885.46    68.5 1877.62   153.3 1859.41   202.2 1844.91   231.6 1833.92
   264.2 1826.03   368.7 1814.21   421.2 1810.53  1499.3 1807.74 1549.881805.785
  1564.9 1803.95  1574.7 1802.88 1589.22 1804.22  1594.4 1808.32  1604.2 1822.86
  1617.3 1834.06    1637 1840.25 1684.561844.829 1809.141851.725 1840.241852.176
 1840.741852.374  1872.9  1861.2 1902.841866.347  1951.6  1874.7  1984.4 1875.96
  1990.9 1878.44    2004 1887.51 2014.871890.839  2108.9 1913.44  2207.2  1944.2
#Mann= 10 ,-1 , 0
       0     .06       0 1549.88     .12       0  1564.9    .045       0
 1589.22     .12       0 1684.56     .06       0 1809.14    .016       0
 1840.24     .08       0 1840.74    .016       0 1902.84     .08       0
 2014.87     .12       0
Bank Sta=1564.9,1589.22
XS Rating Curve= 0 ,0
Exp/Cntr=0.3,0.1

Type RM Length L Ch R = 1 ,24305.3 ,1233.3,1184.2,1184.4
XS GIS Cut Line= 4
     2043797.242      155154.998     2043011.652      155150.658
     2042230.402      155988.332     2042087.173       156435.38
#Sta/Elev= 30
       0 1870.17   137.5 1842.98   199.7 1833.04   376.4 1814.06   464.8 1812.46
   965.6 1810.32    1234 1806.39    1270 1804.54  1616.9 1805.68  1636.5 1804.92
  1652.9 1801.84  1669.2 1801.44  1685.6 1801.97  1711.8  1805.6  1832.9 1807.38
    1859 1809.11  1875.4 1812.68  1901.6 1822.23  1937.6 1832.62  1966.9 1838.43
  2107.1  1856.4 2161.58 1860.51    2169 1858.18  2188.6  1858.4 2200.371861.897
 2207.641864.328  2282.81871.742  2328.8 1874.94 2351.251879.061  2400.5 1884.98
#Mann= 8 ,-1 , 0
       0     .06       0  1652.9    .045       0  1685.6     .06       0
 2161.58    .016       0 2200.37     .08       0 2207.64     .06       0
  2282.8     .08       0 2351.25     .06       0
#XS Ineff= 2 , 0
         1246.47  1819.4
Permanent Ineff=
       F       F
Bank Sta=1652.9,1685.6
XS Rating Curve= 0 ,0
Exp/Cntr=0.3,0.1

Type RM Length L Ch R = 1 ,23121.1 ,566.5,565.7,562.8
XS GIS Cut Line= 3
     2042438.735      154148.054     2041683.527      155597.707
     2041464.923      155765.081
#Sta/Elev= 30
       0 1890.99      59 1875.37    85.2 1866.98   101.6 1856.41   114.6 1850.94
   150.7 1830.82   167.1 1822.59   183.4 1817.19  190.381815.887   216.2  1813.5
   330.8 1810.94   389.8 1811.31   776.3 1806.68   838.6 1804.59     891  1805.1
   956.5    1802   972.9 1802.67   992.5 1799.57  1015.5 1799.58  1028.6 1799.28
    1045 1799.78  1094.1 1803.44  1244.8 1803.29  1516.6 1804.74  1569.1 1806.63
  1631.3 1811.53  1670.6 1815.61  1703.4 1820.22  1752.6 1824.86  1909.9 1836.68
#Mann= 4 ,-1 , 0
       0     .12       0  190.38     .06       0  1015.5    .045       0
    1045     .06       0
Bank Sta=1015.5,1045
XS Rating Curve= 0 ,0
Exp/Cntr=0.3,0.1

Type RM Length L Ch R = 1 ,22555.4 ,693.9,693.8,657.8
XS GIS Cut Line= 2
     2041813.569      154286.945     2041184.395      155745.276
#Sta/Elev= 30
       0 1868.59     9.8 1864.79    26.2 1855.72      72 1827.04    91.7 1816.42
   104.8 1811.03  123.021809.444   189.9 1808.88   248.9 1807.17   684.4 1804.26
   710.6 1802.48   808.9 1802.14     818 1799.07   825.2 1798.56   836.9 1799.23
  840.371800.308   844.9 1801.49   861.3 1802.01   933.3 1801.19   962.8  1803.3
  1224.8 1804.09  1241.1  1805.6  1254.2 1808.29  1267.3 1809.46  1319.7 1817.46
  1391.8 1823.59  1440.9 1829.55  1503.1 1833.21  1539.1 1834.07  1588.3 1837.83
#Mann= 5 ,-1 , 0
       0     .12       0  123.02     .06       0     818    .045       0
   836.9     .12       0  840.37     .06       0
Bank Sta=818,836.9
XS Rating Curve= 0 ,0
Exp/Cntr=0.3,0.1

Type RM Length L Ch R = 1 ,21861.5 ,767.4,760.5,740.1
XS GIS Cut Line= 2
     2041380.902      154055.963     2040698.284      155836.422
#Sta/Elev= 30
       0 1918.87    26.2 1908.29    52.4 1894.78   137.6 1833.04   173.6 1812.44
     190    1806   199.9 1803.92  252.941803.501   635.6 1803.02   701.1 1802.03
  726.851798.599   736.5 1797.67     747 1797.23   753.6 1798.04   763.4 1800.57
   789.6  1799.9  801.831801.613  1087.8 1800.55    1209 1802.73  1474.4 1803.88
  1533.3 1812.57  1569.4 1820.74  1628.3 1830.59  1677.5  1843.4 1694.741851.131
  1713.5 1851.11  1726.6 1858.88 1741.411863.106 1751.511866.868  1906.8  1916.9
#Mann= 9 ,-1 , 0
       0     .12       0  252.94     .06       0  726.85     .12       0
   736.5    .045       0   753.6     .12       0  801.83     .06       0
 1694.74    .016       0 1741.41     .12       0 1751.51     .06       0
#XS Ineff= 2 , 0
          423.97  1822.5
Permanent Ineff=
       F       F
Bank Sta=736.5,753.6
XS Rating Curve= 0 ,0
Exp/Cntr=0.3,0.1

Type RM Length L Ch R = 1 ,21101.1 ,505.4,520.8,532.3
XS GIS Cut Line= 3
     2040906.617       153922.36     2040672.242      154256.561
     2040602.798      155832.082
#Sta/Elev= 30
       0 1878.98   199.2 1876.05   365.7 1899.52   388.6 1901.21   408.2 1899.84
   434.4 1888.32   447.5 1870.27   460.6  1858.6   529.5 1811.34   555.7 1799.79
   585.8 1799.48   827.9 1801.18   870.5 1800.62   903.3 1797.13   913.1 1795.57
   929.5 1796.46  937.451798.964   942.6 1800.56  1060.6 1798.94  1280.3 1802.61
  1519.7 1802.25  1588.5  1803.9  1647.5 1814.65  1732.8 1837.78 1759.811847.855
  1768.8 1852.06  1788.5 1852.65 1805.411862.492 1849.431878.588  1985.2  1925.2
#Mann= 8 ,-1 , 0
       0     .12       0   585.8     .06       0   903.3    .045       0
   929.5     .12       0  937.45     .06       0 1759.81    .016       0
 1805.41     .12       0 1849.43     .06       0
#XS Ineff= 2 , 0
                         1372.53            1828
Permanent Ineff=
       F       F
Bank Sta=903.3,929.5
XS Rating Curve= 0 ,0
Exp/Cntr=0.3,0.1

Type RM Length L Ch R = 1 ,20580.3 ,353.3,359.7,363.3
XS GIS Cut Line= 3
     2040722.806      153998.097     2039815.688      155090.111
       2039676.8      155630.042
#Sta/Elev= 30
       0  1875.8   173.8 1897.09   222.9 1900.03   268.8 1899.98     282 1897.65
   301.6 1889.57   314.8 1879.88   324.6 1868.34   432.8 1799.38   442.6 1797.98
  527.231800.078   566.61800.461   580.3 1800.46   590.2 1795.95   593.4 1795.26
   613.1 1795.67     636 1799.45   704.9 1797.42  731.37 1799.97  1124.6 1801.52
  1547.5 1807.47  1698.4 1817.29  1773.8 1825.32  1794.81829.792 1817.191831.676
  1826.3 1832.34  1839.4 1840.26 1847.691842.742  1895.2 1852.69  1977.1 1875.95
#Mann= 9 ,-1 , 0
       0     .12       0  527.23     .06       0   566.6     .12       0
   590.2    .045       0   613.1     .12       0  731.37     .06       0
  1794.8    .016       0 1817.19     .08       0 1847.69     .06       0
Bank Sta=590.2,613.1
XS Rating Curve= 0 ,0
Exp/Cntr=0.3,0.1

Type RM Length L Ch R = 1 ,20220.6 ,830.5,836.6,820.4
XS GIS Cut Line= 3
     2040719.985      153809.512       2039364.3      155173.445
     2039308.744      155492.889
#Sta/Elev= 30
       0 1855.89    52.4  1856.5   203.1 1876.76   245.7 1881.04   301.4 1883.94
   376.8 1882.16     403 1876.22   422.6 1868.77     439 1859.54   527.4 1802.72
   543.8 1798.93   553.7 1794.78   560.2 1794.35   573.3 1795.15   612.6 1799.59
  767.761799.857  1035.2  1800.5    1566 1808.14    1602 1806.05  1677.4 1806.29
  1752.7 1807.28    1792 1809.65 1925.121811.013 1959.43 1811.16 1989.411811.778
 2016.451810.929  2070.4 1812.03  2090.1 1814.06  2168.7 1829.48  2247.3 1840.99
#Mann= 8 ,-1 , 0
       0     .12       0   553.7    .045       0   573.3     .12       0
  767.76     .06       0 1925.12    .016       0 1959.43     .08       0
 1989.41     .12       0 2016.45     .06       0
Bank Sta=553.7,573.3
XS Rating Curve= 0 ,0
Exp/Cntr=0.3,0.1

Type RM Length L Ch R = 1 ,19384   ,1202.5,1201,1186.6
XS GIS Cut Line= 3
     2040650.541      153722.707     2040316.339       153618.54
     2038753.839      154655.866
#Sta/Elev= 30
       0 1842.89   176.7 1834.18   327.2 1818.34   350.1 1817.58   435.3 1809.02
   474.6 1803.82   563.2 1799.82   602.5 1799.72   615.6 1794.69   635.3 1794.05
   648.4 1795.49   664.8 1799.03  731.611797.812     832 1800.17  1022.2 1798.32
 1136.531799.746 1224.031799.964  1920.6 1803.63  1940.3 1805.72 1952.591811.366
  1973.1 1811.92 1983.341818.095    1996 1825.35 2017.081833.167  2048.5  1843.7
    2078 1851.61    2101 1853.52  2120.6 1860.01  2169.8 1866.27  2225.6 1870.65
#Mann= 9 ,-1 , 0
       0     .12       0   615.6    .045       0   648.4     .12       0
  731.61     .06       0 1136.53    .016       0 1224.03     .06       0
 1952.59    .016       0 1983.34     .12       0 2017.08     .06       0
Bank Sta=615.6,648.4
XS Rating Curve= 0 ,0
Exp/Cntr=0.3,0.1

Type RM Length L Ch R = 1 ,18183   ,1468.4,1477.6,1471
XS GIS Cut Line= 3
     2039962.117      152553.189     2039886.652      152906.735
      2038601.93      154447.533
#Sta/Elev= 30
       0 1959.14   188.9 1904.65   273.6 1890.25   348.5 1873.03   361.5 1871.73
   420.5 1855.05   440.2 1847.72   476.2 1830.69   502.5 1822.58   594.2 1804.88
   623.8 1800.75   630.3 1798.15   636.9 1793.37   646.7 1791.97   669.6 1794.16
   699.1 1797.64  800.461797.113  1207.2 1797.81    1358 1795.69  1489.1 1798.15
  1836.6 1799.46  1925.1 1800.88  1980.8 1803.65  2003.8 1806.54 2012.861809.483
  2039.8  1810.5 2051.241815.311 2101.971828.046    2148 1836.14  2367.6 1850.78
#Mann= 7 ,-1 , 0
       0     .12       0   636.9    .045       0   669.6     .12       0
  800.46     .06       0 2012.86    .016       0 2051.24     .12       0
 2101.97     .06       0
Bank Sta=636.9,669.6
XS Rating Curve= 0 ,0
Exp/Cntr=0.3,0.1

Type RM Length L Ch R = 1 ,16705.4 ,737.2,739,737.3
XS GIS Cut Line= 2
     2039357.138      152377.221     2038254.707      154048.228
#Sta/Elev= 30
       0 1865.54      36 1851.38    85.2 1840.59   193.3 1809.71   239.2 1798.37
   265.4 1796.85  399.751796.844   724.1 1797.35   851.9 1796.23   884.6 1793.07
   893.4 1790.93     901 1790.38   912.5 1791.01   930.5 1795.33  1081.2 1795.15
  1133.6 1793.05  1153.3  1794.9  1251.6 1796.05  1389.2 1793.96  1592.4 1796.76
  1713.6 1802.21  1746.3 1805.99 1767.371810.727  1779.1  1815.5  1795.5 1815.78
 1810.52 1824.05 1850.071834.026  1906.9  1845.4  1959.3 1852.27  2001.9 1854.52
#Mann= 7 ,-1 , 0
       0     .12       0  399.75     .06       0   893.4    .045       0
   912.5     .06       0 1767.37    .016       0 1810.52     .12       0
 1850.07     .06       0
Bank Sta=893.4,912.5
XS Rating Curve= 0 ,0
Exp/Cntr=0.3,0.1

Type RM Length L Ch R = 1 ,15966.4 ,1204.1,1201,1191.3
XS GIS Cut Line= 3
     2038962.173      152099.443     2038128.839      153349.443
     2038033.353      153848.575
#Sta/Elev= 30
       0 1895.71    72.2 1880.68   114.8 1869.43   154.2 1854.28   229.6 1828.13
   275.5 1814.42   298.5 1800.77   308.3 1796.44   321.5 1795.28  545.361796.582
   744.6 1795.67   856.1 1793.11  1131.7 1794.63    1171 1792.41  1180.4 1790.37
  1190.7  1789.7  1197.3 1790.84  1207.1 1794.62  1308.8  1794.2  1364.6 1799.85
  1597.4 1803.77  1676.1 1803.77  1685.9 1802.36 1751.881806.622  1784.3 1807.93
 1798.51  1813.8    1863 1827.62 1897.151833.362 1914.511835.802  2010.5  1844.1
#Mann= 8 ,-1 , 0
       0     .12       0  545.36     .06       0  1180.4    .045       0
  1197.3     .06       0 1751.88    .016       0 1798.51     .06       0
 1897.15     .12       0 1914.51     .06       0
Bank Sta=1180.4,1197.3
XS Rating Curve= 0 ,0
Exp/Cntr=0.3,0.1

Type RM Length L Ch R = 1 ,14765.4 ,2519.1,2530.2,2524.9
XS GIS Cut Line= 3
     2038202.624      151496.144     2037933.527      151687.116
     2037280.966         153729.
#Sta/Elev= 30
       0 1867.13      98 1832.54  243.04 1806.94   362.8 1798.22   536.5 1792.83
   867.5 1793.78   965.8 1791.54  1057.6 1793.61  1083.8 1791.63  1139.6 1793.97
 1212.191793.545 1220.82  1789.1  1231.4 1788.27    1239 1789.07    1251 1792.66
 1286.051792.768 1533.691792.734 1567.411792.331  1844.3 1798.52  1893.4 1801.88
  1926.2 1806.05 1934.161809.015    1959 1811.04 1969.191815.464  1998.3 1820.32
  2116.3  1848.3 2188.871859.214  2309.7 1870.27 2384.531874.234  2473.6 1878.19
#Mann= 12 ,-1 , 0
       0     .12       0  243.04     .06       0 1212.19     .12       0
 1220.82    .045       0    1239     .12       0 1286.05     .06       0
 1533.69     .12       0 1567.41     .06       0 1934.16    .016       0
 1969.19     .12       0 2188.87     .06       0 2384.53     .12       0
#XS Ineff= 2 , 0
                         1646.41         1809.64
Permanent Ineff=
       F       F
Bank Sta=1220.82,1239
XS Rating Curve= 0 ,0
Exp/Cntr=0.3,0.1

Type RM Length L Ch R = 1 ,12235.2 ,1191,1206,1208.8
XS GIS Cut Line= 3
     2037239.082      151400.658      2036262.52        152989.2
     2035928.319      153175.832
#Sta/Elev= 30
       0 1885.69      59 1870.49   104.9 1854.77   140.9 1837.85   216.3 1797.03
   239.2 1792.42  271.911791.161   704.6 1790.28   740.6    1792 1184.981789.638
  1202.7  1786.2  1215.8 1785.81  1226.7 1786.31 1255.081786.361 1269.251786.361
  1294.5 1791.06  1310.9 1791.33    1324 1787.65  1356.8 1791.55    1537 1791.08
  1569.8  1794.9  1704.1 1796.98  1894.2 1809.83 2041.811816.366 2092.481819.666
 2167.521824.538 2176.76 1825.24 2235.191828.846 2237.341828.807  2247.5  1828.9
#Mann= 13 ,-1 , 0
       0     .12       0  271.91     .06       0 1184.98     .12       0
  1202.7    .045       0  1226.7     .06       0 1255.08     .08       0
 1269.25     .06       0 2041.81    .016       0 2092.48     .06       0
 2167.52     .12       0 2176.76     .08       0 2235.19     .06       0
 2237.34     .08       0
#XS Ineff= 2 , 0
                         1387.79         1806.43
Permanent Ineff=
       F       F
Bank Sta=1202.7,1226.7
XS Rating Curve= 0 ,0
Exp/Cntr=0.3,0.1

Type RM Length L Ch R = 1 ,11029.2 ,797.9,806.1,807
XS GIS Cut Line= 4
     2037165.298      151313.853     2036893.076      151387.811
     2035828.492      152186.248     2035533.353      152255.693
#Sta/Elev= 30
       0 1893.11    68.9 1880.21   190.2 1851.59   252.6 1831.03   308.3 1803.89
   331.2  1794.2   350.9 1791.94   403.4 1791.81  427.141789.837   475.5 1791.54
   544.3 1789.01   570.5 1791.28   642.6 1790.67     682    1790   724.3 1785.94
   731.1 1785.04   744.2 1786.26   757.4 1788.96   780.3  1790.4     836 1789.23
   891.7 1790.91   993.3 1790.35  1026.1 1788.92  1065.4 1789.81  1157.2 1788.91
  1468.6 1792.11  1498.1  1795.2  1642.2 1801.02  1694.3  1804.4    1916 1822.97
#Mann= 4 ,-1 , 0
       0     .12       0  427.14     .06       0   724.3    .045       0
   744.2     .06       0
Bank Sta=724.3,744.2
XS Rating Curve= 0 ,0
Exp/Cntr=0.3,0.1

Type RM Length L Ch R = 1 ,10223.1 ,916.4,917.2,904
XS GIS Cut Line= 3
     2036804.744      150980.449     2036034.061       151379.27
     2035461.874      151690.186
#Sta/Elev= 30
       0 1874.75    26.2 1876.66    65.5 1876.82    81.9 1875.46    98.2 1872.61
   157.2 1857.44   189.9 1847.34     203 1842.48   229.2 1829.19   255.4 1812.45
   271.8 1800.24   281.6 1798.08   291.4 1792.46   304.5 1790.75  377.911789.984
   635.3 1788.67   681.1 1789.55   831.7  1789.6  850.221787.275   854.7 1786.16
   864.5 1784.25   875.3    1786   890.7 1789.28  928.891788.853     979 1789.62
  1116.5 1787.83    1231 1789.88  1352.1 1798.69  1404.4  1801.4    1519 1810.57
#Mann= 6 ,-1 , 0
       0     .12       0  377.91     .06       0  850.22     .12       0
   854.7    .045       0   875.3     .12       0  928.89     .06       0
Bank Sta=854.7,875.3
XS Rating Curve= 0 ,0
Exp/Cntr=0.3,0.1

Type RM Length L Ch R = 1 ,9305.9  ,1178.3,1180.9,1180.8
XS GIS Cut Line= 3
     2036390.992      150350.311     2036282.485      150532.603
     2035154.013      151348.575
#Sta/Elev= 30
       0 1923.38    22.8 1917.29      49 1907.75   127.3 1872.81   182.8 1852.39
   225.2 1835.16   261.3 1823.24   300.6 1817.09   320.3 1812.48   336.6 1805.14
     353 1795.51   366.1 1794.38   379.2 1790.92  448.521790.332   621.7 1789.29
   628.3 1788.24   631.6 1785.58   634.8 1783.68   644.7 1783.36     661 1784.66
  668.851786.841     684 1788.16  1073.9 1788.57  1254.1 1787.17  1267.2 1788.27
  1290.2 1794.84 1312.291798.518    1395 1810.68  1499.9 1822.26  1604.7 1829.69
#Mann= 7 ,-1 , 0
       0     .12       0  448.52     .06       0   631.6    .045       0
     661     .08       0  668.85     .06       0 1312.29     .08       0
    1395     .06       0
Bank Sta=631.6,661
XS Rating Curve= 0 ,0
Exp/Cntr=0.3,0.1

Type RM Length L Ch R = 1 ,8125    ,371.1,367.2,362.6
XS GIS Cut Line= 3
     2035828.492      149933.644      2035789.43      150102.915
      2034530.54      150918.519
#Sta/Elev= 30
       0  1908.4    19.7 1901.67    39.3 1893.65    49.2 1888.51    68.8 1876.38
    91.8 1860.35   104.9 1848.74   121.3 1837.61   160.6 1812.21   173.7 1804.49
   183.5 1800.22   203.2  1794.2   239.2 1790.09  341.041789.064   805.8  1788.7
   900.8    1787   959.8 1787.65   979.4 1787.36   989.2 1784.08   995.8 1782.39
  1015.4 1781.97  1020.1 1783.21  1028.5 1786.26  1041.6 1786.24  1051.4 1787.88
  1071.1 1793.71  1126.8 1805.58  1208.7 1819.83    1284 1827.35  1673.7 1857.61
#Mann= 4 ,-1 , 0
       0     .12       0  341.04     .06       0   989.2    .045       0
  1020.1     .06       0
Bank Sta=989.2,1020.1
XS Rating Curve= 0 ,0
Exp/Cntr=0.3,0.1

Type RM Length L Ch R = 1 ,7757.9  ,517.7,519.6,519
XS GIS Cut Line= 4
     2035494.291      149668.887     2035289.885      149951.597
     2034734.742      150393.714     2034417.902       150497.88
#Sta/Elev= 30
       0 1860.88    39.1 1846.25    52.2 1843.48    78.2 1834.65   104.3 1829.26
     150 1821.69   198.9 1816.17   270.6 1803.03  391.941794.331   466.6 1787.37
   708.6 1787.35     774 1786.49   796.9 1784.73   801.7 1783.23   816.5 1782.01
   826.4  1782.1   832.9 1783.37   842.7 1786.82   855.8 1786.65   862.3 1787.69
   904.8 1801.82   940.8 1810.78     967 1816.22 1029.991826.275 1044.381828.438
    1137 1838.54 1266.211849.266    13561856.412 1367.491857.265  1392.1 1858.94
#Mann= 9 ,-1 , 0
       0     .12       0  391.94     .06       0   801.7    .045       0
   832.9     .06       0 1029.99     .08       0 1044.38     .06       0
 1266.21     .08       0    1356     .06       0 1367.49     .08       0
Bank Sta=801.7,832.9
XS Rating Curve= 0 ,0
Exp/Cntr=0.3,0.1

Type RM Length L Ch R = 1 ,7238.3  ,628.4,627.1,620.3
XS GIS Cut Line= 3
     2035312.867      149224.443     2034526.409      149979.651
     2034344.117      150344.235
#Sta/Elev= 30
       0 1918.37     108 1899.02   196.5 1885.97   255.4  1874.5   311.1  1861.8
   343.8 1857.12     478 1821.85   517.3 1809.56  543.45 1803.17  574.311798.098
   605.8 1792.78   628.7 1786.67  683.37  1786.4   707.2  1786.7   730.2 1783.78
   749.8  1785.2   756.4 1783.58   759.6 1782.37   772.7 1781.96   783.1 1782.95
   795.7 1784.77   825.1 1785.43   841.5 1787.23   949.6 1820.95  1018.3 1832.62
  1116.4 1840.51 1431.19 1857.49 1461.751858.819 1485.121859.739    1498 1860.07
#Mann= 9 ,-1 , 0
       0     .12       0  543.45     .06       0  574.31     .12       0
  683.37     .06       0   756.4    .045       0   783.1     .06       0
 1431.19     .08       0 1461.75     .06       0 1485.12     .08       0
Bank Sta=756.4,783.1
XS Rating Curve= 0 ,0
Exp/Cntr=0.3,0.1

Type RM Length L Ch R = 1 ,6611.2  ,386.3,388.1,388.4
XS GIS Cut Line= 2
      2034826.31      148820.923     2033982.602       149918.69
#Sta/Elev= 30
       0    1924    26.2 1919.22   176.8 1883.27   261.8 1857.28   274.9 1852.65
   333.9 1839.58   369.9 1829.26  388.771825.905   477.9 1813.61   513.9 1806.53
   582.6 1794.84   621.9 1786.84   644.8 1783.71   661.2 1783.95   677.1 1781.45
     707 1781.28   716.8  1781.7  721.651782.305   733.2 1784.07   752.8 1784.28
   782.3 1786.64   821.6 1791.98  848.091796.868   864.1 1799.25  894.471801.993
  1017.9  1819.6  1037.6 1823.02  1191.4 1843.29  1289.6 1854.39  1384.5 1863.63
#Mann= 7 ,-1 , 0
       0     .12       0  388.77     .06       0   677.1    .045       0
   716.8     .08       0  721.65     .06       0  848.09     .12       0
  894.47     .06       0
Bank Sta=677.1,716.8
XS Rating Curve= 0 ,0
Exp/Cntr=0.3,0.1
